--- LaurCk.prj (project) ---

Proj Title=LaurCk
Current Plan=p01
Default Exp/Contr=0,0
English Units
Geom File=g01
Flow File=f01
Plan File=p01
BEGIN DESCRIPTION:
END DESCRIPTION:
DSS Export Rating Curves= 0
DSS Export Rating Curve Sorted= 0
DSS Export Volume Flow Curves= 0
DXF OffsetX= 0
DXF OffsetY= 0
DXF ScaleX= 0
DXF ScaleY= 0

--- LaurCk.p01 (plan) ---

Plan Title=Floodplain
Program Version=4.00
Geom File=g01
Flow File=f01
K Sum by GR=0
Std Step Tol=0.01
Critical Tol=0.01
Num of Std Step Trials=20
Max Error Tol=0.3
Flow Tol Ratio=0.001
Split Flow NTrial=30
Split Flow Tol=0.02
Split Flow Ratio=0.02
Log Output Level=0
Friction Slope Method=1
Unsteady Friction Slope Method=2
Unsteady Bridges Friction Slope Method=1
Global Log Level=0
CheckData=False
Run HTab=0
Run UNet=0
Run PostProcess=0
UNET Theta=0
UNET Theta Warmup=0
UNET ZTol=0
UNET ZSATol=0
UNET MxIter=0
UNET MaxInSteps=0
UNET DtIC=0
UNET DtMin=0
UNET MaxCRTS=0
UNET WFStab=0
UNET SFStab=0
UNET WFX=0
UNET SFX=0
UNET DSS MLevel=0
UNET DZMax Abort=0
UNET Convert EG Bridges=0
UNET Use Existing IB Tables=0
UNET Froude Limit=0
UNET Froude Power=0
Write IC File=0
Echo Input=False
Echo Output=False
Write Detailed=0

--- LaurCk.f01 (steady flow) ---

Flow Title=NFF Regression Equation
Program Version=4.00
Number of Profiles=1
Profile Names=P100yr
River Rch & RM=LaurCk,Main      ,42625.2
531.5361
River Rch & RM=LaurCk,Main      ,42107
590.3180
River Rch & RM=LaurCk,Main      ,39175.6
651.5766
River Rch & RM=LaurCk,Main      ,38939.5
722.8619
River Rch & RM=LaurCk,Main      ,36580.7
760.6633
River Rch & RM=LaurCk,Main      ,36252.2
945.0779
River Rch & RM=LaurCk,Main      ,30856.5
1017.338
River Rch & RM=LaurCk,Main      ,30362.1
1532.993
River Rch & RM=LaurCk,Main      ,29843.1
1536.145
River Rch & RM=LaurCk,Main      ,29307.7
1926.233
River Rch & RM=LaurCk,Main      ,28251.2
1941.107
River Rch & RM=LaurCk,Main      ,23420.7
2156.639
River Rch & RM=LaurCk,Main      ,23249.5
2554.575
River Rch & RM=LaurCk,Main      ,22563.5
2817.655
River Rch & RM=LaurCk,Main      ,19540.1
2986.984
River Rch & RM=LaurCk,Main      ,19151.7
3334.310
River Rch & RM=LaurCk,Main      ,8232.9
3700.646
River Rch & RM=LaurCk,Main      ,5894.3
4106.242
River Rch & RM=LaurCk,Main      ,3243.4
4331.440
River Rch & RM=LaurCk,Main      ,146.1
4792.349
Boundary for River Rch & Prof#=LaurCk,Main      ,1
Up Type=0
Dn Type=3
Dn Slope=0.005146

--- LaurCk.g01 (geometry) ---

Geom Title=USGS 10m DEM
Program Version=4.10

River Reach=LaurCk          ,Main
Reach XY= 30
      2110103.94      394749.726     2109411.651      395623.885
     2109300.559      397909.499     2107929.871      400629.082
     2107615.347      400645.789     2106284.611      402020.108
     2105248.786      402522.766     2104581.516      403942.657
     2103427.237      404185.265     2102166.384      405603.241
     2102150.929      406194.387     2100671.208      407572.858
     2099982.052      409138.006     2098695.291      410224.124
     2097607.515      410688.419     2096616.531      413340.205
     2096079.432      413918.224     2096326.126      414766.087
     2095329.768      415303.386     2095435.443      416686.621
     2094857.935      417911.641     2094163.891      418268.376
     2093271.852      419267.928     2090580.558      419755.904
     2089642.739      420188.673     2089725.084      421223.477
      2088949.21      422246.386     2087985.878      422298.304
     2088238.605      423419.147     2087799.968      423856.007

Type RM Length L Ch R = 1 ,42625.2 ,270.2,264.9,259.6
XS GIS Cut Line= 2
     2109791.706      394426.076     2110410.952      395101.349
#Sta/Elev= 30
       0 3450.45    10.1 3447.85    30.2 3440.74    40.3 3437.97    50.3 3436.41
    80.6 3434.96   161.1 3422.98   251.7 3412.57   312.1 3406.24   412.8 3397.51
   433.13394.795     443 3393.58   453.1 3393.25   463.1 3394.89   483.3 3400.48
   503.4 3403.16   513.5 3403.62   543.7 3403.52   614.2 3407.38   644.4 3409.97
   664.5 3412.71   674.6  3414.6   694.7 3419.91   714.8 3426.98   785.3 3450.43
   795.4 3453.11   825.6 3457.04   835.7  3458.8   845.7 3461.47   916.2 3485.52
#Mann= 3 , 0 , 0
       0      .1       0   433.1    .045       0   463.1      .1       0
Bank Sta=433.1,463.1
XS Rating Curve= 0 ,0
Exp/Cntr=0.3,0.1

Type RM Length L Ch R = 1 ,42360.3 ,246.5,253.3,260.2
XS GIS Cut Line= 2
     2109623.352      394756.905     2110308.701      395218.689
#Sta/Elev= 30
       0 3481.26    50.4 3460.02   110.9  3435.1   171.3 3409.57   181.4 3405.94
   191.5 3404.07   201.6 3403.08   292.3 3396.36   322.5 3393.35   332.6 3391.79
   355.63386.128   362.8 3384.61   372.9 3384.32   385.63386.085   403.1 3390.09
   463.6  3401.6   503.9 3410.04   594.6 3423.96   624.8 3428.12   634.9 3430.67
     645 3434.37   675.2 3447.12   685.3 3451.08   695.4 3454.46   705.5 3456.96
   715.6 3458.04   745.8 3459.25   755.9 3460.02   765.9 3462.13   826.4  3485.9
#Mann= 3 , 0 , 0
       0      .1       0   355.6    .045       0   385.6      .1       0
Bank Sta=355.6,385.6
XS Rating Curve= 0 ,0
Exp/Cntr=0.3,0.1

Type RM Length L Ch R = 1 ,42107   ,327.7,315,302.2
XS GIS Cut Line= 2
      2109510.79      394830.573      2110029.33      395474.051
#Sta/Elev= 30
       0 3511.07    50.4 3487.67    80.6 3473.93   181.4 3429.67   221.7 3412.33
   231.8  3408.4   241.9 3405.53   272.1 3399.27   312.4 3390.48   332.6 3386.29
   342.7 3384.73   352.7 3383.91     383 3382.94     393 3382.39   403.1 3381.45
   411.23380.351   423.3 3378.92   433.4 3378.79   441.23380.031   443.4 3380.38
   463.6 3386.89   473.7 3388.16   503.9 3389.51   584.5 3393.89   594.6 3394.63
   614.8 3397.44   655.1 3403.82   685.3 3409.11   765.9 3425.71   826.4 3437.78
#Mann= 3 , 0 , 0
       0      .1       0   411.2    .045       0   441.2      .1       0
Bank Sta=411.2,441.2
XS Rating Curve= 0 ,0
Exp/Cntr=0.3,0.1

Type RM Length L Ch R = 1 ,41792.2 ,216.4,220.3,224.2
XS GIS Cut Line= 2
     2109198.492      395206.919     2109968.245      395507.631
#Sta/Elev= 30
       0 3513.57    50.4 3491.06   120.9 3461.01   141.1 3452.86   201.6 3429.01
     262 3404.51   272.1 3400.71   282.2 3397.41   322.5 3385.17   342.7 3379.56
   352.7 3377.16   372.9 3373.05     383 3371.46   386.63371.158     393 3370.62
   403.1 3370.84   416.63372.468   433.4 3374.45   453.5 3376.23   524.1 3379.46
   544.2 3380.56   574.4 3382.85   594.6 3384.97   634.9  3391.3   665.2 3395.37
   715.6 3403.02   755.9 3410.46     776 3414.43   796.2  3418.8   826.4 3425.71
#Mann= 3 , 0 , 0
       0      .1       0   386.6    .045       0   416.6      .1       0
Bank Sta=386.6,416.6
XS Rating Curve= 0 ,0
Exp/Cntr=0.3,0.1

Type RM Length L Ch R = 1 ,41571.7 ,472.9,469,465.1
XS GIS Cut Line= 3
     2109140.527      395340.099     2109533.097       395579.46
     2109921.919      395824.206
#Sta/Elev= 30
       0 3505.14      10  3499.9      20 3495.21      50 3481.77      80 3467.36
   129.9 3444.21   209.9 3405.81   239.9 3392.08   249.9 3388.26   259.9 3385.02
   299.9 3373.66   309.9  3370.9   319.8 3368.72   329.8 3367.71   369.8 3365.93
   379.8 3364.85   388.73363.141   399.8 3361.28   409.8 3361.28   418.73363.024
   429.8    3366   439.8 3367.93   449.8 3368.66   479.8 3369.26   509.7 3371.02
   649.6 3381.58   659.5 3383.08   749.4 3401.34   829.3 3414.45   919.2 3430.27
#Mann= 3 , 0 , 0
       0      .1       0   388.7    .045       0   418.7      .1       0
Bank Sta=388.7,418.7
XS Rating Curve= 0 ,0
Exp/Cntr=0.3,0.1

Type RM Length L Ch R = 1 ,41102.7 ,276,275.8,275.9
XS GIS Cut Line= 3
     2108948.089      395797.999     2109374.693      395969.505
     2109798.486       396146.94
#Sta/Elev= 30
       0 3456.69      30 3440.96      80 3415.59   119.9 3396.25   139.9 3387.06
   159.9 3378.87   229.9 3356.77   239.9 3354.25   249.9  3352.3   279.9 3348.45
   369.8 3345.14   389.8 3344.04   399.8  3342.6   422.43337.574   429.8 3336.56
   439.8 3336.53   452.43337.552   499.7 3341.58   539.7 3345.93   549.7 3347.76
   559.7 3351.09   579.6 3359.02   599.6 3365.62   669.5 3386.58   699.5 3396.08
   709.5 3398.92   719.5 3400.99   769.4 3407.41   859.3 3416.75   919.2 3423.59
#Mann= 3 , 0 , 0
       0      .1       0   422.4    .045       0   452.4      .1       0
Bank Sta=422.4,452.4
XS Rating Curve= 0 ,0
Exp/Cntr=0.3,0.1

Type RM Length L Ch R = 1 ,40826.9 ,297,287.2,277.2
XS GIS Cut Line= 3
     2108845.928      396044.217     2109268.563      396214.128
     2109688.411      396389.911
#Sta/Elev= 30
       0 3450.01    49.5 3430.84   128.7 3401.75     198 3378.52   277.3 3353.21
   297.1 3348.13   366.4 3336.56   386.2 3334.06   415.9 3332.23   425.8 3329.87
   435.7 3325.84   440.53324.623   445.6 3323.33   455.5  3323.9   470.53327.433
   485.2  3330.8     505 3333.21   603.9 3337.88   623.7 3339.36   633.6 3341.26
   742.5 3373.41   791.9 3390.38   801.8 3392.39   811.7 3392.72   821.6 3391.75
   831.5  3391.9   841.4 3394.09   851.3 3397.06   861.2 3399.09   910.7 3404.71
#Mann= 3 , 0 , 0
       0      .1       0   440.5    .045       0   470.5      .1       0
Bank Sta=440.5,470.5
XS Rating Curve= 0 ,0
Exp/Cntr=0.3,0.1

Type RM Length L Ch R = 1 ,40539.6 ,300,298.4,296.7
XS GIS Cut Line= 3
     2108715.563       396524.55      2109165.89      396495.931
     2109616.228       396473.75
#Sta/Elev= 30
       0 3444.39    40.1 3424.68    60.2 3415.61   110.3 3397.06   140.4 3380.29
   150.4 3375.77   180.5  3366.7   220.6 3353.01   250.7 3345.75   300.8 3336.02
   340.9 3327.17   441.2 3318.59   461.2 3314.98   489.23307.888   501.3 3305.44
   511.4 3305.38   519.23307.159   541.4 3314.81   551.4 3316.77   651.6 3324.75
   671.7 3326.69   681.7 3328.38   711.8 3338.08   731.8 3342.06   741.8 3345.41
   761.8 3355.33   781.9 3363.13     852 3384.59   872.1 3388.84   902.1  3393.3
#Mann= 3 , 0 , 0
       0      .1       0   489.2    .045       0   519.2      .1       0
Bank Sta=489.2,519.2
XS Rating Curve= 0 ,0
Exp/Cntr=0.3,0.1

Type RM Length L Ch R = 1 ,40241.3 ,265.8,269.8,273.8
XS GIS Cut Line= 2
     2108807.604      396841.638     2109726.069        396729.1
#Sta/Elev= 30
       0 3411.16    30.2 3394.37    50.3 3384.06    80.5 3370.08   120.7 3353.35
   140.8 3345.68     171 3335.11   241.4 3313.25   271.6 3303.42   281.6 3300.86
   291.7 3299.74     342 3297.67   382.2 3296.62   422.4 3293.14   434.1 3291.13
   442.6 3289.49   452.6 3289.24   464.13291.857   472.7 3294.48   482.8 3296.84
   502.9 3300.37     523 3302.86   603.5 3311.08   653.8 3320.28   724.2 3339.88
   774.5 3354.68   814.7 3367.47     865 3384.58   885.1 3389.72   925.3 3396.62
#Mann= 3 , 0 , 0
       0      .1       0   434.1    .045       0   464.1      .1       0
Bank Sta=434.1,464.1
XS Rating Curve= 0 ,0
Exp/Cntr=0.3,0.1

Type RM Length L Ch R = 1 ,39971.4 ,280.8,282.7,284.7
XS GIS Cut Line= 2
     2108850.608      397030.622        2109775.      397072.372
#Sta/Elev= 30
       0 3401.86    30.2 3385.09    50.3 3372.53    70.4 3360.85    90.5 3351.31
   110.6 3343.95     171 3323.89   281.6 3285.53   291.7 3282.42   301.7  3280.3
   311.8 3279.21   372.2  3274.9   382.2 3272.29   400.93263.941   402.3 3263.34
   412.4 3262.23   422.4  3263.8   430.93266.122   452.6    3272   462.7  3273.9
   472.7  3275.1   583.4 3281.98   593.4    3283   603.5 3284.87   643.7 3297.02
   724.2 3323.26   754.4 3332.33   834.8 3354.78   854.9  3359.1   925.3 3370.06
#Mann= 3 , 0 , 0
       0      .1       0   400.9    .045       0   430.9      .1       0
Bank Sta=400.9,430.9
XS Rating Curve= 0 ,0
Exp/Cntr=0.3,0.1

Type RM Length L Ch R = 1 ,39688.6 ,224,221.5,219
XS GIS Cut Line= 2
     2108887.095      397256.955     2109803.339       397386.34
#Sta/Elev= 30
       0 3384.37    20.1 3373.59    60.4 3353.69    80.5 3342.78    90.5 3338.17
   120.7 3325.88   221.3 3288.72   291.7 3260.44   301.7 3257.11   321.9 3253.04
     342  3248.3     352 3245.62   372.2 3239.07   378.23237.558   382.2 3236.55
   392.3 3237.21   408.23244.636   412.4 3246.74   422.4 3249.45   432.5 3250.09
   462.7 3249.44   492.8 3250.41     513 3251.48   563.2 3255.29   583.4 3257.64
   633.6  3265.7   663.8 3271.09   744.3 3287.81   854.9 3317.05   925.3 3333.01
#Mann= 3 , 0 , 0
       0      .1       0   378.2    .045       0   408.2      .1       0
Bank Sta=378.2,408.2
XS Rating Curve= 0 ,0
Exp/Cntr=0.3,0.1

Type RM Length L Ch R = 1 ,39467.2 ,292.6,291.6,290.5
XS GIS Cut Line= 2
     2108860.017      397510.375     2109784.945      397537.786
#Sta/Elev= 30
       0 3380.28    30.2 3366.64    50.3 3358.32   150.9 3322.17   191.1 3307.01
   211.2 3298.72   221.3 3293.84   241.4 3282.87   271.6 3264.86   311.8 3238.91
   321.9 3231.85   331.9 3224.22   335.1 3222.36     342 3218.35     352 3216.69
   365.13217.986   442.6 3226.62   492.8 3232.89   502.9 3233.55   533.1  3233.7
   543.1  3234.2   553.2 3235.04   593.4 3240.11   663.8 3245.37   673.9 3247.33
   704.1 3255.49   734.2 3262.59   814.7 3279.83   885.1 3294.31   925.3 3301.24
#Mann= 3 , 0 , 0
       0      .1       0   335.1    .045       0   365.1      .1       0
Bank Sta=335.1,365.1
XS Rating Curve= 0 ,0
Exp/Cntr=0.3,0.1

Type RM Length L Ch R = 1 ,39175.6 ,226.5,236.1,245.6
XS GIS Cut Line= 2
     2108896.216      397803.004     2109821.392      397785.912
#Sta/Elev= 30
       0 3315.17    40.2 3305.41    80.5 3293.57   221.3 3249.43   291.7 3229.46
   311.8 3221.44   321.9 3217.94     342 3212.39   385.43202.052   392.3 3200.59
   402.3 3199.98   412.4 3203.06   415.43205.007   422.4 3209.55   432.5 3213.53
   442.6 3214.57   452.6 3215.16   482.8 3218.53   502.9 3219.74   533.1 3217.56
   553.2 3218.47   593.4 3221.85   653.8 3229.44     694 3236.76   744.3 3247.59
   764.4 3253.68   804.6 3267.42   824.8  3272.6   885.1 3282.35   925.3 3287.48
#Mann= 3 , 0 , 0
       0      .1       0   385.4    .045       0   415.4      .1       0
Bank Sta=385.4,415.4
XS Rating Curve= 0 ,0
Exp/Cntr=0.3,0.1

Type RM Length L Ch R = 1 ,38939.5 ,284.1,284.2,284.2
XS GIS Cut Line= 2
     2108828.385       397839.25     2109681.511      398197.606
#Sta/Elev= 30
       0 3321.31    30.2 3313.06   110.6 3287.48   160.9 3269.02   211.2  3249.2
   241.4 3239.64   281.6 3229.33   301.7 3225.79     352 3218.53   362.1 3216.64
   372.2 3213.55   392.3 3204.02   412.4    3193     4223190.273   432.5 3190.14
   442.6 3192.02     4523194.558   462.7 3196.91   472.7 3197.92   563.2 3200.85
   573.3 3201.75   583.4  3204.6   593.4 3209.59   613.5 3222.02   623.6 3226.72
   633.6 3229.92   704.1 3248.55   754.4  3264.7   854.9 3298.56   925.3  3326.1
#Mann= 3 , 0 , 0
       0      .1       0     422    .045       0     452      .1       0
Bank Sta=422,452
XS Rating Curve= 0 ,0
Exp/Cntr=0.3,0.1

Type RM Length L Ch R = 1 ,38655.4 ,367.2,372.8,378.4
XS GIS Cut Line= 2
      2108695.37      398089.021     2109548.497      398447.376
#Sta/Elev= 30
       0 3308.66    40.2 3298.19    50.3 3295.22   140.8 3266.56   191.1 3251.74
   241.4 3238.46     342 3213.23   412.4 3190.44   432.5 3183.17   436.33182.139
   442.6 3180.43   452.6 3179.81   462.7 3181.23   466.33182.101   482.8 3185.49
   492.8 3185.93   573.3 3186.21   613.5 3185.79   623.6 3187.68   633.6    3193
   653.8 3207.72   673.9 3222.96   704.1 3247.16   714.1 3254.06   724.2 3258.66
   764.4 3269.06   784.5 3274.86   885.1 3307.83   905.2 3315.04   925.3 3322.93
#Mann= 3 , 0 , 0
       0      .1       0   436.3    .045       0   466.3      .1       0
Bank Sta=436.3,466.3
XS Rating Curve= 0 ,0
Exp/Cntr=0.3,0.1

Type RM Length L Ch R = 1 ,38282.5 ,281.8,280.3,278.9
XS GIS Cut Line= 2
     2108638.065      398338.023     2109379.687      398891.412
#Sta/Elev= 30
       0 3272.35    60.4 3254.94    90.5 3247.14   211.2 3219.76   261.5 3210.49
   301.7 3199.75   331.9 3194.46   382.2 3189.97   392.3 3188.03   432.5  3175.2
   442.6 3171.52   453.73166.663   462.7 3163.25   472.7 3162.11   483.73163.377
     513 3167.03   533.1 3170.36   553.2  3174.3   573.3 3179.72   593.4 3187.61
   623.6  3201.9   673.9 3224.18     694  3232.5   714.1 3239.33   724.2 3242.16
   764.4 3251.94   784.5  3257.8   834.8 3278.84   905.2 3306.28   925.3 3313.22
#Mann= 3 , 0 , 0
       0      .1       0   453.7    .045       0   483.7      .1       0
Bank Sta=453.7,483.7
XS Rating Curve= 0 ,0
Exp/Cntr=0.3,0.1

Type RM Length L Ch R = 1 ,38002.2 ,326.1,318.3,310.2
XS GIS Cut Line= 2
      2108461.52      398584.507     2109250.598      399102.402
#Sta/Elev= 30
       0 3279.68    20.1 3273.24    50.2 3259.88    70.3 3252.01   130.5 3231.13
   230.9 3193.71   261.1 3183.58   281.2 3177.87   291.2 3175.76   301.2 3174.65
   401.6 3168.25   411.7 3166.82   441.8 3159.53   493.63148.293     502 3147.79
   512.1 3149.58   523.63154.456   542.2 3163.14   572.3    3175   612.5 3192.08
   622.5 3194.84   662.7 3202.67   682.8  3205.5   712.9 3208.44   773.2 3218.98
   793.2 3225.16   823.4 3235.88   853.5 3245.28   913.7 3268.24   943.8 3277.26
#Mann= 3 , 0 , 0
       0      .1       0   493.6    .045       0   523.6      .1       0
Bank Sta=493.6,523.6
XS Rating Curve= 0 ,0
Exp/Cntr=0.3,0.1

Type RM Length L Ch R = 1 ,37683.9 ,186.8,181.1,175.6
XS GIS Cut Line= 2
     2108220.912      398963.107     2109138.719       399183.31
#Sta/Elev= 30
       0 3310.72    50.2 3285.71   110.4 3254.18   140.6 3239.01   170.7 3225.81
   230.9 3201.58   271.1 3186.68   311.3 3173.31   321.3 3170.38   401.6 3150.59
   411.7 3147.69   427.1 3142.38   431.8 3140.86   442.1 3139.21   451.8 3139.09
   522.1 3144.12   532.2  3145.7   552.2 3150.47   562.3    3152   572.3 3152.62
   612.5 3152.62   642.6 3155.65   662.7 3159.14   692.8 3166.69     723 3175.59
   793.2 3198.92   833.4 3210.87   873.6 3223.81   913.7 3236.95   943.8 3247.36
#Mann= 3 , 0 , 0
       0      .1       0   427.1    .045       0   442.1      .1       0
Bank Sta=427.1,442.1
XS Rating Curve= 0 ,0
Exp/Cntr=0.3,0.1

Type RM Length L Ch R = 1 ,37502.8 ,265.1,276.6,289.1
XS GIS Cut Line= 2
     2108227.261      399245.246     2109170.981       399229.37
#Sta/Elev= 30
       0 3265.71    50.2 3241.28    80.3  3227.9   110.4 3216.75   180.7 3193.93
   200.8  3185.9     251 3163.87   271.1 3156.11   291.2 3150.56   331.4 3142.09
   351.4  3137.2   371.5 3134.01   381.6 3133.78   396.3 3133.87   411.3  3134.3
   461.9 3140.01     502 3143.08   522.1 3143.63   542.2 3142.88   552.2 3143.41
   572.3  3146.3   602.5 3151.79   682.8 3168.26   712.9 3176.02     743 3185.58
   813.3 3215.24   833.4 3222.77   853.5 3229.34   893.6 3240.81   943.8 3257.56
#Mann= 3 , 0 , 0
       0      .1       0   396.3    .045       0   411.3      .1       0
Bank Sta=396.3,411.3
XS Rating Curve= 0 ,0
Exp/Cntr=0.3,0.1

Type RM Length L Ch R = 1 ,37226.2 ,385.7,387,387.4
XS GIS Cut Line= 3
     2108210.269      399291.744     2108617.118      399510.247
     2109006.259      399743.702
#Sta/Elev= 30
       0 3267.46    50.2 3244.55    80.3 3231.34   130.5 3210.46   150.6 3202.94
   160.6 3199.59   180.7 3193.32   230.9 3178.84   381.5 3133.47   391.5 3130.71
   401.6 3128.68   444.63124.394   451.8 3123.71   461.8 3123.34   474.63124.313
   492.1 3127.07   502.2 3127.85   522.3 3128.86   542.5 3129.37     603 3128.99
   683.7 3125.76   693.8 3125.58   703.8 3126.28   713.9  3128.5   744.2 3137.55
   764.3 3142.73   784.5 3147.15   814.8 3153.06   824.8 3155.49   915.6 3180.41
#Mann= 3 , 0 , 0
       0      .1       0   444.6    .045       0   474.6      .1       0
#XS Ineff= 2 , 0
                          552.65         3129.41
Permanent Ineff=
       F       F
Bank Sta=444.6,474.6
XS Rating Curve= 0 ,0
Exp/Cntr=0.3,0.1

Type RM Length L Ch R = 1 ,36839.2 ,254.6,258.5,262.4
XS GIS Cut Line= 3
     2108107.163      399646.034       2108488.1      399880.967
     2108850.837        400129.2
#Sta/Elev= 30
       0 3256.24    49.7  3233.2    99.5  3211.4   109.4 3207.92   248.6 3167.21
   268.5 3160.08   288.4 3147.86   328.2 3118.81   338.2 3113.12   348.1 3109.86
   390.83106.448   407.8 3105.79   420.83105.939   457.6 3106.17   487.5 3107.92
   497.5 3109.91   507.5 3113.08   527.5 3121.19   547.4 3128.21   567.4 3132.65
   577.4 3133.52   637.4 3136.02   677.3 3135.99   687.3 3134.71   707.3 3129.75
   727.3  3126.4   747.2 3124.91   767.2  3124.7   807.2 3125.95   887.1 3131.34
#Mann= 3 , 0 , 0
       0      .1       0   390.8    .045       0   420.8      .1       0
Bank Sta=390.8,420.8
XS Rating Curve= 0 ,0
Exp/Cntr=0.3,0.1

Type RM Length L Ch R = 1 ,36580.7 ,326.4,328.5,330.6
XS GIS Cut Line= 3
      2108004.48      399808.143     2108340.446      400103.835
     2108656.233      400409.574
#Sta/Elev= 30
       0 3243.14    39.8 3221.75    69.6 3204.96    79.6    3200    89.5 3196.21
   119.4 3186.05   139.2 3177.42     179 3157.94   228.8 3135.51   288.4 3103.39
   298.4  3100.1   308.3 3099.07   349.83099.074   379.83098.979   397.8 3098.47
   457.6 3101.82   537.5 3104.55   557.4 3106.15   567.4 3108.84   587.4 3115.55
   597.4 3118.42   607.4 3120.72   627.4 3124.15   657.3 3127.62   727.3 3133.39
   757.2 3134.76   767.2 3135.93   777.2 3137.86   827.2 3149.48   887.1 3167.24
#Mann= 3 , 0 , 0
       0      .1       0   349.8    .045       0   379.8      .1       0
Bank Sta=349.8,379.8
XS Rating Curve= 0 ,0
Exp/Cntr=0.3,0.1

Type RM Length L Ch R = 1 ,36252.2 ,666.9,667.4,667.9
XS GIS Cut Line= 2
     2107767.903      399975.881      2108425.11      400663.721
#Sta/Elev= 30
       0 3253.62      30 3236.25    50.1 3226.89   150.2 3186.83   210.3 3164.71
   280.4 3137.95   320.4 3123.76   340.5  3118.8   370.5 3113.88   380.5 3111.14
   390.6 3106.76   400.6 3101.69     4263087.818   430.6 3085.55   440.6 3083.36
   450.6 3082.91     4563083.364   460.6 3083.75   470.7 3086.24   490.7 3092.47
   500.7 3093.69   520.7 3094.81   600.8 3093.62   670.9 3090.21     681  3091.3
     691 3094.96   841.2 3177.84   851.2 3182.89   871.2 3192.01   951.3 3225.34
#Mann= 3 , 0 , 0
       0      .1       0     426    .045       0     456      .1       0
Bank Sta=426,456
XS Rating Curve= 0 ,0
Exp/Cntr=0.3,0.1

Type RM Length L Ch R = 1 ,35584.8 ,476.1,475.1,466.7
XS GIS Cut Line= 2
     2107353.426      400317.863     2108010.632      401005.704
#Sta/Elev= 30
       0 3220.13      30 3208.62   100.1 3183.31   130.2 3173.96   170.2 3162.69
   200.3 3151.19   290.4 3113.68   310.4 3106.68   340.5 3099.12   350.5 3095.43
   390.6 3077.76   409.63070.741   420.6 3068.17   430.6 3067.72   439.63068.521
   470.7 3074.45   490.7 3076.28   500.7 3077.89   510.7 3081.15   520.7 3085.88
   530.8 3089.28   540.8 3091.79   580.8 3098.65   610.9  3105.4   650.9  3116.8
     731  3142.3   751.1  3150.4   851.2  3197.2   861.2 3201.35   951.3 3234.78
#Mann= 3 , 0 , 0
       0      .1       0   409.6    .045       0   439.6      .1       0
Bank Sta=409.6,439.6
XS Rating Curve= 0 ,0
Exp/Cntr=0.3,0.1

Type RM Length L Ch R = 1 ,35109.7 ,423.4,422.6,429.3
XS GIS Cut Line= 2
     2107062.728      400597.527     2107719.935      401285.368
#Sta/Elev= 30
       0 3211.25      30 3197.26   100.1 3168.59   180.2 3139.48   270.4 3104.43
   300.4  3094.2   320.4 3086.73   380.5  3063.1   393.23057.824   400.6 3054.76
   410.6 3053.19   420.6 3054.14   423.23054.972   440.6 3060.28   450.6 3062.37
   460.6 3063.59   470.7 3064.01   530.8  3064.9   570.8 3066.66   580.8 3068.13
   590.8 3071.97   600.8 3077.57   630.9 3095.56   650.9  3106.6     731 3145.91
   751.1 3155.43   791.1 3171.49   841.2 3190.71   911.3 3214.68   951.3 3229.02
#Mann= 3 , 0 , 0
       0      .1       0   393.2    .045       0   423.2      .1       0
Bank Sta=393.2,423.2
XS Rating Curve= 0 ,0
Exp/Cntr=0.3,0.1

Type RM Length L Ch R = 1 ,34687   ,457.9,461,464
XS GIS Cut Line= 2
     2106779.423      400858.044      2107436.63      401545.884
#Sta/Elev= 30
       0 3207.35    80.1 3169.47   120.2  3152.7   200.3  3120.7   220.3 3111.98
   230.3 3106.73   320.4 3054.38   330.5 3050.93   340.5 3049.92   400.6 3048.17
   410.6  3046.9   420.6 3044.04   427.53041.308   430.6 3040.08   440.6 3038.32
   450.6 3038.84   457.53040.317   480.7 3046.66   490.7 3050.68   530.8 3069.39
   540.8 3073.07   580.8 3085.17   610.9  3095.1     691 3123.09     721 3134.13
   761.1 3147.56   821.2 3165.65   861.2 3181.44   931.3 3206.98   951.3  3213.5
#Mann= 3 , 0 , 0
       0      .1       0   427.5    .045       0   457.5      .1       0
Bank Sta=427.5,457.5
XS Rating Curve= 0 ,0
Exp/Cntr=0.3,0.1

Type RM Length L Ch R = 1 ,34226.1 ,405.6,402.3,399
XS GIS Cut Line= 2
     2106471.242      401114.097     2107023.854      401868.583
#Sta/Elev= 30
       0 3217.99    90.5 3173.03   130.7 3153.66   251.4 3107.31   271.5 3098.27
   341.9 3064.69   372.1 3051.68   382.1 3047.94   392.2 3044.87   432.4 3033.58
   450.33026.914   462.6 3022.81   472.6 3022.38   480.33023.897   492.8  3027.1
   502.8 3027.76   593.3  3023.5   603.4 3023.32   613.4 3025.28   623.5 3030.84
   633.5 3038.22   643.6 3046.37   653.6 3053.21   663.7 3058.16   703.9 3072.36
     724 3080.08   774.3 3102.86   804.5 3115.16   844.7 3129.98   935.2 3161.29
#Mann= 3 , 0 , 0
       0      .1       0   450.3    .045       0   480.3      .1       0
#XS Ineff= 2 , 0
                          503.99         3027.63
Permanent Ineff=
       F       F
Bank Sta=450.3,480.3
XS Rating Curve= 0 ,0
Exp/Cntr=0.3,0.1

Type RM Length L Ch R = 1 ,33823.8 ,380.3,388.4,396.5
XS GIS Cut Line= 2
     2106072.801      401361.839     2106727.887       402029.29
#Sta/Elev= 30
       0  3226.4    80.4 3191.45   120.7 3176.02   130.7 3170.96   150.8  3159.2
     171 3149.99   221.2 3128.93   241.4 3119.79   291.6 3095.07   341.9 3071.62
   432.4 3027.43   462.6 3011.48   466.93009.868   472.6 3007.73   482.7  3006.9
   496.93009.281   512.9 3012.54     533 3015.47   573.2 3018.09   613.4 3019.43
   623.5 3020.84   663.7 3029.99   693.9 3033.52   703.9 3035.53     714 3038.41
     724 3042.25   754.2 3056.07   794.4 3071.75   864.8 3098.13   935.2 3123.57
#Mann= 3 , 0 , 0
       0      .1       0   466.9    .045       0   496.9      .1       0
Bank Sta=466.9,496.9
XS Rating Curve= 0 ,0
Exp/Cntr=0.3,0.1

Type RM Length L Ch R = 1 ,33435.3 ,248.7,249.2,249.6
XS GIS Cut Line= 2
     2106056.914       401620.01     2106444.492      402471.135
#Sta/Elev= 30
       0 3124.75   160.9 3062.99   251.4 3031.64   261.5 3029.51   271.5 3028.41
   341.9 3023.89     362 3021.85   372.1  3019.8   392.2 3014.47   422.4 3005.59
   446.2 2997.62   452.5 2995.56   462.6 2994.17   476.22995.535   492.8 2997.21
     543 2995.84   553.1 2997.72   563.1 3002.43   583.2 3015.77   623.5 3046.27
   643.6 3060.68   653.6 3066.96   673.8 3077.08   683.8 3081.15   703.9  3088.1
   764.3 3106.36   834.7 3126.21   864.8 3135.35     895 3142.96   935.2 3155.34
#Mann= 3 , 0 , 0
       0      .1       0   446.2    .045       0   476.2      .1       0
Bank Sta=446.2,476.2
XS Rating Curve= 0 ,0
Exp/Cntr=0.3,0.1

Type RM Length L Ch R = 1 ,33186.7 ,216.7,210.6,204.5
XS GIS Cut Line= 2
     2105838.072       401712.95      2106225.65      402564.074
#Sta/Elev= 30
       0 3153.87    20.1 3145.47    80.4 3118.43   160.9 3084.78   271.5 3039.89
   311.7 3021.86   331.8  3014.7   341.9 3011.84   392.2 2999.56   424.32988.328
   432.4  2986.7   442.5 2987.07   454.32989.248   462.6 2990.76   472.6 2991.32
   522.9 2989.57     533 2990.01     543 2992.54   553.1 2997.42   593.3 3022.67
   603.4 3028.27   613.4 3032.01   653.6 3040.81   703.9 3054.16   744.2 3066.57
   814.5 3086.54   834.7 3093.28   864.8 3104.32   874.9 3107.42   935.2 3122.76
#Mann= 3 , 0 , 0
       0      .1       0   424.3    .045       0   454.3      .1       0
Bank Sta=424.3,454.3
XS Rating Curve= 0 ,0
Exp/Cntr=0.3,0.1

Type RM Length L Ch R = 1 ,32975.5 ,357.7,364.6,371.4
XS GIS Cut Line= 2
     2105583.424      401900.453     2106165.996      402632.053
#Sta/Elev= 30
       0 3142.72    30.2 3130.25    70.4 3112.63    90.5 3103.22   130.7 3083.19
   150.8  3074.6   160.9 3070.75   241.4 3042.61   281.6  3027.3   341.9 3006.42
   402.2  2987.3   437.82979.007   442.5 2978.16   452.5  2977.6   462.6 2978.84
   467.82980.161   492.8 2987.05   502.8 2990.57   512.9 2994.62     533  3004.1
     543 3008.09   553.1 3010.96   633.5 3026.94   663.7 3032.39   673.8 3035.02
   683.8  3038.4   703.9 3046.34   764.3 3072.15   804.5 3088.61   935.2 3130.21
#Mann= 3 , 0 , 0
       0      .1       0   437.8    .045       0   467.8      .1       0
Bank Sta=437.8,467.8
XS Rating Curve= 0 ,0
Exp/Cntr=0.3,0.1

Type RM Length L Ch R = 1 ,32610.9 ,372.8,367.2,357.8
XS GIS Cut Line= 3
     2105410.542       402038.93     2105584.943      402469.501
     2105752.542      402900.507
#Sta/Elev= 30
       0  3116.8    29.6  3105.4    79.1 3089.64    98.8 3082.79   247.1 3028.33
   286.6 3014.64   296.5 3010.42   306.4 3005.15   345.9 2982.65   355.8  2977.8
   365.7 2975.36   375.6 2974.86   405.2 2975.62     425 2974.94   454.7 2971.28
   481.42967.273   484.7 2966.95   494.7 2967.81   511.42972.344   524.9 2975.24
     555 2976.62   575.1 2978.92   595.2 2982.96   615.4 2988.42   635.4 2995.22
   695.8 3019.29     746 3040.57   776.2 3051.72   836.5 3072.16     927 3097.78
#Mann= 3 , 0 , 0
       0      .1       0   481.4    .045       0   511.4      .1       0
Bank Sta=481.4,511.4
XS Rating Curve= 0 ,0
Exp/Cntr=0.3,0.1

Type RM Length L Ch R = 1 ,32243.8 ,475.6,458.6,441.8
XS GIS Cut Line= 3
     2105020.092      402151.454     2105257.994      402550.465
      2105489.24      402950.941
#Sta/Elev= 30
       0 3155.61     9.9 3156.66    39.5 3154.73    59.3 3152.68    79.1 3148.75
   118.6 3136.53   158.1 3122.06   177.9  3113.5   207.6  3097.4   296.5  3043.5
   306.4 3035.59   316.3 3025.91   345.9 2994.55   355.8 2985.82   365.7  2978.5
   375.6  2972.6   385.5    2968   405.2 2961.32   424.52956.597   434.9 2955.94
   454.52958.702   474.6  2962.9   494.7 2964.43   524.9  2963.7   685.7 2963.68
   725.9 2964.43     736 2966.28     746 2969.32   856.6 3007.47     927 3030.57
#Mann= 3 , 0 , 0
       0      .1       0   424.5    .045       0   454.5      .1       0
Bank Sta=424.5,454.5
XS Rating Curve= 0 ,0
Exp/Cntr=0.3,0.1

Type RM Length L Ch R = 1 ,31785.2 ,369.7,373.7,377.4
XS GIS Cut Line= 3
     2104684.209      402817.011     2105119.863      402965.779
     2105551.411      403119.918
#Sta/Elev= 30
       0 3138.41      20 3128.65    80.1 3103.31   120.1 3085.26   160.1 3066.08
   270.2 3011.17   350.3 2974.61   370.3 2966.92   410.3 2954.59   430.3 2946.92
     4362945.506   440.3 2944.44   450.4 2944.16     4662946.208   480.3 2947.74
     560    2953   579.9 2954.75   609.8 2959.83   619.8 2962.49   629.7 2966.19
   639.7 2970.57   679.5 2988.73   719.4  3004.7   769.2 3026.36   789.1 3034.62
     809 3042.22   858.8 3060.31   888.7 3071.97   898.7 3075.42   918.6 3080.81
#Mann= 3 , 0 , 0
       0      .1       0     436    .045       0     466      .1       0
Bank Sta=436,466
XS Rating Curve= 0 ,0
Exp/Cntr=0.3,0.1

Type RM Length L Ch R = 1 ,31411.5 ,288.4,288.4,288.4
XS GIS Cut Line= 3
     2104558.717      403085.946     2104959.303      403304.147
     2105354.964      403526.896
#Sta/Elev= 30
       0 3129.19     9.9 3125.44    29.8  3117.2    59.5 3104.33    99.2 3086.38
   138.8 3068.12     238 3023.44   247.9  3018.1   257.8 3012.34   297.5 2987.56
   317.3 2975.47   337.2 2964.12   366.9 2947.88   386.7 2935.57   390.92933.978
   396.7 2931.78   406.6 2931.69   420.92933.314   426.4 2933.97   436.3 2934.56
   446.2 2934.72   526.8 2935.58   617.6 2935.93   627.7 2936.18   637.8 2937.59
   647.9 2940.31     668 2947.43   819.4 3004.71   859.8 3020.76   910.2 3041.83
#Mann= 3 , 0 , 0
       0      .1       0   390.9    .045       0   420.9      .1       0
Bank Sta=390.9,420.9
XS Rating Curve= 0 ,0
Exp/Cntr=0.3,0.1

Type RM Length L Ch R = 1 ,31123.1 ,256.1,266.6,277
XS GIS Cut Line= 3
      2104401.94      403328.726     2104802.526      403546.926
     2105198.187      403769.676
#Sta/Elev= 30
       0 3080.21    49.6 3066.22    79.3 3058.69   138.8 3045.02   168.6  3040.3
   178.5 3037.85   208.2 3028.43   228.1 3023.04     238 3019.42   267.8 3006.18
   317.3 2982.18   366.9 2959.91   376.8 2954.45   386.7 2947.92   406.6 2932.39
   417.72925.292   426.4 2922.04   436.3  2921.9   447.72923.469   466.2 2925.81
   486.4 2926.88   627.7 2929.12   688.2 2931.61   708.4 2933.05   718.5 2934.89
   738.7 2940.18   799.2 2957.78   859.8 2974.74   879.9 2979.19   910.2 2983.62
#Mann= 3 , 0 , 0
       0      .1       0   417.7    .045       0   447.7      .1       0
Bank Sta=417.7,447.7
XS Rating Curve= 0 ,0
Exp/Cntr=0.3,0.1

Type RM Length L Ch R = 1 ,30856.5 ,485.2,494.4,501.2
XS GIS Cut Line= 2
     2104394.836        403432.2     2104950.788      404152.628
#Sta/Elev= 30
       0 3043.79      40 3033.02      70 3024.24     110 3010.79     140 2999.74
     200 2975.26     230 2962.34     250 2952.53     290 2931.99     300 2927.17
     310 2923.27     320 2921.03     360 2920.96   411.32917.329     430 2915.65
     440 2915.29   441.32915.312     460 2915.92     520 2919.49     550 2920.86
     580 2921.62     660 2922.77     740 2924.78     760 2925.97     770 2927.23
     780 2929.13     790 2931.91     850 2951.72     880 2960.14     910  2967.5
#Mann= 3 , 0 , 0
       0      .1       0   411.3    .045       0   441.3      .1       0
Bank Sta=411.3,441.3
XS Rating Curve= 0 ,0
Exp/Cntr=0.3,0.1

Type RM Length L Ch R = 1 ,30362.1 ,518,519,519.9
XS GIS Cut Line= 3
     2104122.479      403504.499     2104287.894      403928.365
      2104453.31      404352.231
#Sta/Elev= 30
       0 2982.37    19.8 2976.24    69.2 2965.03   108.8 2954.42   148.4 2942.45
   197.8 2926.67   237.4  2913.5   247.3 2911.86   257.2  2911.6   326.4  2911.6
   346.2 2911.26   385.8  2907.8   412.22904.966   425.3 2903.95   434.7 2903.88
   442.22904.177   534.1 2909.47     544 2911.13   553.9 2914.74   593.5 2935.83
   692.4 2985.03   702.3 2989.54   712.2 2993.24     732 2999.18   751.7 3005.91
   781.4 3018.03   811.1 3032.06   850.6 3052.11   890.2 3069.55     910 3078.85
#Mann= 3 , 0 , 0
       0      .1       0   412.2    .045       0   442.2      .1       0
Bank Sta=412.2,442.2
XS Rating Curve= 0 ,0
Exp/Cntr=0.3,0.1

Type RM Length L Ch R = 1 ,29843.1 ,545.3,535.4,525.6
XS GIS Cut Line= 2
     2103640.879      403659.786     2103971.711      404507.519
#Sta/Elev= 30
       0 2948.63      40 2940.45      70 2931.92     120  2914.3     150 2901.99
     160 2899.44     170 2898.93     230 2898.63     320 2900.42   434.82895.412
   464.82894.199     470  2894.1     480 2894.89     490 2898.13     500 2905.57
     510 2914.81     520 2923.21     530 2930.24     540 2936.16     550 2940.79
     560 2944.23     580 2949.87     610 2960.08     630 2967.74     650 2976.19
     690 2995.04     870 3088.35     880 3092.69     890 3096.08     910 3100.73
#Mann= 3 , 0 , 0
       0      .1       0   434.8    .045       0   464.8      .1       0
Bank Sta=434.8,464.8
XS Rating Curve= 0 ,0
Exp/Cntr=0.3,0.1

Type RM Length L Ch R = 1 ,29307.7 ,465.6,460.4,455.1
XS GIS Cut Line= 3
     2102961.559      403897.714     2103278.778      404215.883
     2103622.496      404559.536
#Sta/Elev= 30
       0 3038.86    79.9 3000.91   149.8  2968.5   169.7 2959.67   219.6  2941.2
   269.6 2923.32   309.5 2909.79   329.5  2903.5   339.5 2900.76   369.4 2894.19
   379.4 2892.17   389.4 2890.72   399.4 2889.77   439.3  2887.2   508.8 2883.42
   518.7 2883.14     5292883.446     5592886.592     608  2891.2   617.9 2893.39
   627.8  2897.8   647.7 2910.88   677.4 2929.16   687.4    2935   697.3 2939.63
     737 2951.04   766.7 2960.04   796.5 2969.47   895.6 3002.22   935.3 3016.36
#Mann= 3 , 0 , 0
       0      .1       0     529    .045       0     559      .1       0
Bank Sta=529,559
XS Rating Curve= 0 ,0
Exp/Cntr=0.3,0.1

Type RM Length L Ch R = 1 ,28847.3 ,258.5,258.6,258.6
XS GIS Cut Line= 3
     2102582.998      404347.165     2102964.129      404584.167
     2103376.882      404839.925
#Sta/Elev= 30
       0 2991.07      10 2987.02    49.9  2972.6    69.8 2966.39   129.7 2948.71
   149.6    2942   169.6 2933.52   219.4 2910.64   239.4 2902.27   259.3 2894.69
   289.2 2884.45   309.2 2876.82   319.2  2875.4   329.1 2875.22   547.9 2878.01
   557.8 2877.76   583.9 2875.24   587.5 2874.96   597.4  2875.4   607.4 2879.18
   613.92883.428   627.2 2892.08   676.7  2920.7   686.6 2925.97   696.6  2930.3
   746.1 2946.13   785.7 2959.48   825.4 2973.22   904.6 3001.61   934.4    3012
#Mann= 3 , 0 , 0
       0      .1       0   583.9    .045       0   613.9      .1       0
Bank Sta=583.9,613.9
XS Rating Curve= 0 ,0
Exp/Cntr=0.3,0.1

Type RM Length L Ch R = 1 ,28588.7 ,334.8,337.5,340.3
XS GIS Cut Line= 3
     2102417.224      404540.956     2102797.685       404779.93
     2103209.682      405037.802
#Sta/Elev= 30
       0 2995.01    39.9  2976.1    99.8 2951.75   159.8 2928.14   179.7 2921.89
   259.6 2899.56   299.5  2888.9   339.5  2878.9   379.4 2871.64   389.4 2870.22
   419.3 2870.14   469.1 2868.96   498.9 2869.86   548.5 2874.03   558.4 2874.12
   568.3 2873.49   578.82872.309   588.2 2871.19   598.1  2870.6     608 2871.74
   608.82872.136   617.9 2876.64   637.8 2891.48   647.7 2897.88   667.5 2909.76
   687.4 2920.36   697.3 2924.33   707.2 2927.77   756.8 2944.53   935.3 3006.42
#Mann= 3 , 0 , 0
       0      .1       0   578.8    .045       0   608.8      .1       0
Bank Sta=578.8,608.8
XS Rating Curve= 0 ,0
Exp/Cntr=0.3,0.1

Type RM Length L Ch R = 1 ,28251.2 ,308.6,306.1,303.5
XS GIS Cut Line= 3
     2102257.003      404745.607     2102605.498      405029.174
     2102982.991      405335.342
#Sta/Elev= 30
       0  2981.2      30 2969.54   179.7 2913.96   239.6 2893.11   249.6 2890.17
   259.6 2888.49   279.6 2887.19   289.5 2885.73   349.4  2870.8   359.4 2869.01
   369.4 2868.14   459.2 2865.75   512.72862.941   528.6 2862.58   538.6  2863.5
   542.72864.303   558.4 2867.46   588.2 2872.58   627.8  2877.4   637.8 2878.92
   647.7 2881.51   657.6 2885.36   667.5 2889.94   687.4 2899.57   717.1 2914.61
     727 2918.81   816.3 2953.31   875.8 2977.22   915.5 2992.76   935.3 3001.24
#Mann= 3 , 0 , 0
       0      .1       0   512.7    .045       0   542.7      .1       0
Bank Sta=512.7,542.7
XS Rating Curve= 0 ,0
Exp/Cntr=0.3,0.1

Type RM Length L Ch R = 1 ,27945.1 ,542,539,535.9
XS GIS Cut Line= 3
     2102040.166      405024.364     2102420.626      405263.339
     2102832.623       405521.21
#Sta/Elev= 30
       0 2952.11      30 2945.49    59.9 2941.92    79.9 2938.81    99.8 2933.99
   109.8 2930.57   139.8  2918.6   159.8 2912.74   189.7 2905.12   219.6 2899.02
   249.6 2891.52   269.6 2888.52   289.5 2887.51   309.5 2884.92   349.4 2876.74
   359.4 2873.44   369.4 2868.19   379.4 2862.06   389.4 2859.05   399.4 2858.68
   449.3 2860.42   508.8 2861.27   578.2 2860.53   607.72858.815   617.9 2859.31
   637.72864.232   677.4 2874.68   766.7 2904.86   816.3 2923.37   935.3 2970.85
#Mann= 3 , 0 , 0
       0      .1       0   607.7    .045       0   637.7      .1       0
Bank Sta=607.7,637.7
XS Rating Curve= 0 ,0
Exp/Cntr=0.3,0.1

Type RM Length L Ch R = 1 ,27406.1 ,556.6,564.1,571.6
XS GIS Cut Line= 2
     2101478.955      405354.641     2102997.439      406051.401
#Sta/Elev= 30
       0 3125.09    40.3 3106.91   100.6 3083.31   231.5 3037.54   301.9 3010.74
   362.3  2985.4     463 2947.13   563.6 2903.63   664.3 2856.15   674.3 2852.98
   684.4 2851.49   717.22849.008   747.22850.352     785 2854.38   805.2 2855.11
   905.8 2849.25  1056.8 2846.72  1076.9 2848.73  1107.1 2856.35  1117.2 2860.13
  1227.9 2913.78  1258.1 2924.85  1348.6  2946.2  1419.1 2956.14  1449.3 2961.98
  1469.4 2968.05  1509.7 2984.44  1529.8 2990.33  1630.4 3001.73  1670.7 3008.47
#Mann= 3 , 0 , 0
       0      .1       0   717.2    .045       0   747.2      .1       0
#XS Ineff= 2 , 0
                          803.54         2855.26
Permanent Ineff=
       F       F
Bank Sta=717.2,747.2
XS Rating Curve= 0 ,0
Exp/Cntr=0.3,0.1

Type RM Length L Ch R = 1 ,26842   ,432.2,432.2,432.2
XS GIS Cut Line= 2
     2101468.037      405585.549      2102693.23      406721.405
#Sta/Elev= 30
       0 3116.17    30.2 3104.91   110.7 3068.87   181.2 3046.52   201.3 3038.69
   221.4 3029.57   271.7 3004.51   291.9 2995.73   362.3  2970.5   483.1 2930.64
   503.2 2922.95   533.4 2906.79   634.1 2849.83   644.1 2844.67   654.2 2841.29
   674.3 2840.19   899.22839.433   905.8 2839.42   929.22840.206  1006.4 2850.01
  1046.7 2851.24  1066.8 2853.72  1076.9 2855.86    1097 2861.45  1127.2 2871.43
  1197.7 2890.26  1318.4 2924.01  1449.3 2956.12    1560 2979.44  1670.7 3007.76
#Mann= 3 , 0 , 0
       0      .1       0   899.2    .045       0   929.2      .1       0
Bank Sta=899.2,929.2
XS Rating Curve= 0 ,0
Exp/Cntr=0.3,0.1

Type RM Length L Ch R = 1 ,26409.8 ,559.2,563.9,568.7
XS GIS Cut Line= 2
     2101176.136      405851.524     2102401.329       406987.38
#Sta/Elev= 30
       0 3156.81    40.3 3150.98    70.4 3142.19    90.6 3133.52     161 3096.02
   211.4 3073.67   372.4  3016.9   513.3 2957.66   603.9 2924.45   664.3 2896.13
   744.8 2851.64     785 2832.84   794.82830.133   805.2 2829.54   824.82830.025
   986.3 2833.98  1026.6 2831.16  1056.8 2832.62  1066.8 2835.09    1087  2845.5
  1167.5 2891.66  1187.6 2900.71  1308.4 2944.11  1358.7 2956.54  1449.3 2983.69
  1489.6 3001.11  1519.7 3022.63  1529.8 3027.11  1610.3 3049.22  1670.7 3070.73
#Mann= 3 , 0 , 0
       0      .1       0   794.8    .045       0   824.8      .1       0
Bank Sta=794.8,824.8
XS Rating Curve= 0 ,0
Exp/Cntr=0.3,0.1

Type RM Length L Ch R = 1 ,25845.9 ,275.1,271.1,266.7
XS GIS Cut Line= 2
     2100972.962      406219.043      2101972.36      407557.875
#Sta/Elev= 30
       0 3002.84    40.3 2986.81    60.4 2980.14    80.5 2975.46     151 2963.08
   201.3 2949.91   261.7 2931.92   352.3 2900.08   533.4 2831.01   553.6 2824.97
   573.7 2823.99   674.3 2824.13   744.8 2820.45   754.8 2819.98   774.82821.135
   825.3 2824.06   865.6 2824.27   875.6 2825.71   885.7  2830.5   925.9 2860.08
   956.1 2879.52   976.3 2891.53   996.4 2901.06  1107.1 2934.31    1248 2978.73
  1348.6 3022.86    1409 3045.56  1479.5 3063.49  1570.1 3088.24  1670.7 3108.88
#Mann= 3 , 0 , 0
       0      .1       0   744.8    .045       0   774.8      .1       0
#XS Ineff= 2 , 0
          672.23 2824.26  836.47         2824.53
Permanent Ineff=
       F       F
Bank Sta=744.8,774.8
XS Rating Curve= 0 ,0
Exp/Cntr=0.3,0.1

Type RM Length L Ch R = 1 ,25574.8 ,322.3,318,313.7
XS GIS Cut Line= 2
      2100585.29      406405.089     2101854.604      407491.417
#Sta/Elev= 30
       0 2903.67    60.4 2900.74     161 2887.72   191.2 2880.65   221.4  2869.3
   241.6 2863.22   271.7 2858.97   362.3 2857.72   452.9 2850.99   503.2  2849.1
   573.7 2841.34   664.3 2822.22     785 2821.78   795.1 2821.34   810.12818.254
   825.3 2815.27   835.4 2815.01   840.1 2815.17   976.3 2823.51   996.4 2827.01
  1016.5 2834.84  1036.6  2847.3  1066.8 2868.95    1087 2879.61  1187.6 2911.08
  1258.1 2937.56  1479.5 3016.26  1529.8 3030.37  1610.3  3049.6  1670.7 3069.66
#Mann= 3 , 0 , 0
       0      .1       0   810.1    .045       0   840.1      .1       0
Bank Sta=810.1,840.1
XS Rating Curve= 0 ,0
Exp/Cntr=0.3,0.1

Type RM Length L Ch R = 1 ,25256.8 ,559.9,559.2,557.8
XS GIS Cut Line= 2
     2100393.623      406803.514     2102274.823      407947.714
#Sta/Elev= 30
       0 3026.19    70.4  3002.1   110.6 2992.04   160.9  2981.8     191  2972.4
   261.4 2939.69   311.7 2919.93   462.5 2851.82   512.8 2828.07   542.9 2811.14
     553 2809.88   653.5 2816.37   723.9 2818.02   794.3 2814.31     8312809.759
   844.5  2809.1   854.6 2811.59     8612814.777   884.8 2825.52   995.4 2865.43
  1075.8 2897.11  1196.4 2938.47  1407.6 3008.38  1588.5 3057.58  1658.9 3090.63
  1769.5 3129.06  2030.9 3190.17  2101.3 3209.01  2161.6 3218.03  2201.8 3221.92
#Mann= 3 , 0 , 0
       0      .1       0     831    .045       0     861      .1       0
#XS Ineff= 2 , 0
          723.12 2818.03
Permanent Ineff=
       F       F
Bank Sta=831,861
XS Rating Curve= 0 ,0
Exp/Cntr=0.3,0.1

Type RM Length L Ch R = 1 ,24697.6 ,684.5,680.9,677.9
XS GIS Cut Line= 2
     2100158.222      407278.572     2102066.052      408377.796
#Sta/Elev= 30
       0 3043.91    80.4 3010.98     181 2964.31   291.6 2919.29   351.9 2897.41
   422.3 2876.91   542.9 2816.69   573.1 2798.96   576.52798.073   593.2 2795.88
   606.52796.339   683.7 2803.36     925 2803.14     935 2806.11   995.4 2835.34
  1015.5 2847.68  1045.6 2869.49  1095.9 2889.97  1176.3 2915.88  1367.4 2972.72
  1528.2 3028.93  1578.5 3042.61    1669 3064.08  1739.4 3083.13  1809.7 3092.18
  1880.1    3097  2020.9 3102.78  2101.3 3099.38  2161.6 3106.41  2201.8 3107.24
#Mann= 3 , 0 , 0
       0      .1       0   576.5    .045       0   606.5      .1       0
Bank Sta=576.5,606.5
XS Rating Curve= 0 ,0
Exp/Cntr=0.3,0.1

Type RM Length L Ch R = 1 ,24016.4 ,587.6,595.6,603.7
XS GIS Cut Line= 2
     2099873.596      407973.759     2101928.346      408765.029
#Sta/Elev= 30
       0 2951.49    90.5 2931.89   201.1 2905.12     372 2856.69   392.1 2849.75
   532.9  2789.6   545.12785.699     553 2784.69   575.1 2786.66   623.4 2791.51
   864.6 2788.66   945.1 2789.47  1005.4 2791.87  1025.5 2794.83  1156.2 2826.08
  1216.5 2834.76  1246.7 2843.28  1266.8 2847.21  1437.7 2866.36    1488 2873.91
  1558.4 2886.55  1648.9 2896.98  1699.1 2899.14  1779.6 2905.86    1860 2905.46
  1920.3 2907.88  1960.5 2911.31    2041 2922.41  2141.5 2922.16  2201.8 2927.02
#Mann= 3 , 0 , 0
       0      .1       0   545.1    .045       0   575.1      .1       0
#XS Ineff= 2 , 0
                          625.63         2791.48
Permanent Ineff=
       F       F
Bank Sta=545.1,575.1
XS Rating Curve= 0 ,0
Exp/Cntr=0.3,0.1

Type RM Length L Ch R = 1 ,23420.7 ,167,171.2,175.4
XS GIS Cut Line= 2
     2099875.332      408421.625     2101563.544      409835.149
#Sta/Elev= 30
       0  2870.4   201.1 2815.22   331.8 2776.86   341.8 2775.53   445.62773.357
   462.5 2773.03   475.62773.326   583.1 2779.47   643.5  2780.7   723.9 2780.41
   754.1 2782.97   794.3 2790.78   824.4 2798.51   844.5 2806.93   874.7 2823.08
   884.8 2827.41   955.1 2854.41  1015.5 2875.58  1035.6 2879.49  1156.2 2897.99
  1196.4 2900.48  1367.4 2903.06  1417.6 2905.65  1518.2 2912.89  1638.8 2925.19
  1729.3 2932.34  1870.1 2941.07  1930.4 2946.85  2010.8 2952.98  2201.8 2976.07
#Mann= 3 , 0 , 0
       0      .1       0   445.6    .045       0   475.6      .1       0
Bank Sta=445.6,475.6
XS Rating Curve= 0 ,0
Exp/Cntr=0.3,0.1

Type RM Length L Ch R = 1 ,23249.5 ,687,686,685
XS GIS Cut Line= 2
     2099839.011      408516.218     2100639.007      409443.432
#Sta/Elev= 30
       0  2862.4    30.1 2853.44    40.2 2849.96    90.3 2830.34   110.4    2823
   120.5 2820.03     261 2784.92   291.1 2776.04   301.1 2774.33   341.3 2773.52
   431.6 2770.46   440.52770.645   470.52773.199     522 2776.49     542 2777.08
   722.7  2776.8     793 2778.14     803 2778.89   813.1 2780.83   873.3 2797.41
   883.3 2799.61   903.4 2803.25   913.4 2804.57   933.5 2805.99   973.7 2806.37
    1044 2808.15  1124.2  2808.3  1164.4 2807.76  1204.6 2805.74  1224.6 2805.42
#Mann= 3 , 0 , 0
       0      .1       0   440.5    .045       0   470.5      .1       0
Bank Sta=440.5,470.5
XS Rating Curve= 0 ,0
Exp/Cntr=0.3,0.1

Type RM Length L Ch R = 1 ,22563.5 ,350.9,351.1,351.3
XS GIS Cut Line= 2
     2099360.541      408975.526     2100122.951      409825.822
#Sta/Elev= 30
       0 2882.68      30 2874.72    40.1 2871.65    70.1 2861.05   110.2 2846.42
   150.3 2831.19   240.4 2796.21   280.5 2781.98   310.6 2772.84   350.6 2762.54
   360.6 2760.27   370.7 2758.91   380.7 2758.64     4212760.137     4512761.543
   460.8 2762.67   490.9 2767.45   500.9  2768.4   681.2 2770.95   691.2 2771.16
   701.3 2772.48   711.3 2774.98   721.3  2778.1   801.4  2804.4   961.7 2860.28
  1031.8 2882.67  1051.9  2888.7  1071.9 2893.88    1122 2903.84    1142 2908.48
#Mann= 3 , 0 , 0
       0      .1       0     421    .045       0     451      .1       0
Bank Sta=421,451
XS Rating Curve= 0 ,0
Exp/Cntr=0.3,0.1

Type RM Length L Ch R = 1 ,22212.4 ,397.9,392.9,388
XS GIS Cut Line= 2
     2099070.873      409175.425     2099804.005      409993.067
#Sta/Elev= 30
       0 2876.87    40.3 2862.37    80.6 2847.05   100.8  2839.7   191.4 2808.89
   211.6 2801.12   241.8 2789.01   302.2 2764.12   312.3 2761.73   322.4 2760.75
   382.9  2757.6   433.2 2754.62   442.12754.682   453.4 2755.25   472.12756.934
   513.8 2760.27     534 2761.42   755.6 2760.87   765.7 2761.21   775.8 2763.24
   785.9 2767.65   795.9 2772.66     806 2777.78   826.2 2788.75   836.2 2793.52
   876.5  2810.4   906.8 2822.66  1057.9 2881.67    1078 2888.95  1098.2  2895.4
#Mann= 3 , 0 , 0
       0      .1       0   442.1    .045       0   472.1      .1       0
Bank Sta=442.1,472.1
XS Rating Curve= 0 ,0
Exp/Cntr=0.3,0.1

Type RM Length L Ch R = 1 ,21819.4 ,297.7,310.7,323.6
XS GIS Cut Line= 2
     2098802.743      409582.946      2099550.66      410101.328
#Sta/Elev= 30
       0 2787.81      30 2786.98      60 2785.77      80 2785.36     150  2781.9
     160 2780.98     170 2779.25     180 2776.84     210 2768.76     240 2761.06
     250 2758.81     260 2757.19     330 2747.82     340 2747.03   347.92747.046
   377.92749.483     440 2754.47     460 2755.51     500  2755.7     660 2755.03
     670 2755.22     680 2756.05     690 2757.68     700 2760.46     710 2763.85
     730 2771.57     810 2804.71     840 2816.47     860 2823.28     910 2838.93
#Mann= 3 , 0 , 0
       0      .1       0   347.9    .045       0   377.9      .1       0
Bank Sta=347.9,377.9
XS Rating Curve= 0 ,0
Exp/Cntr=0.3,0.1
